--- RamonaFlowControl.prj (project) ---

Proj Title=Ramona Flow Control Rating Curve
Current Plan=p05
Default Exp/Contr=0.3,0.1
English Units
Geom File=g05
Flow File=f04
Plan File=p05
Y Axis Title=Elevation
X Axis Title(PF)=Main Channel Distance
X Axis Title(XS)=Station
BEGIN DESCRIPTION:
San Jacinto River Alternatives Analysis - Alternative 5
W.O. 03-461  jcc  May 2007
This model is made up of the following Plans:
END DESCRIPTION:
DSS File=..\..\..\..\..\2003\03-0461\hyd\Alternative 5\HEC-RAS\SJRalt5.dss
DSS Export Rating Curves= 0
DSS Export Rating Curve Sorted= 0
DSS Export Volume Flow Curves= 0
DXF Filename=..\..\..\..\..\2003\03-0461\hyd\Alternative 5\HEC-RAS\SJRalt5.
DXF OffsetX= 0
DXF OffsetY= 0
DXF ScaleX= 1
DXF ScaleY= 10

--- RamonaFlowControl.p05 (plan) ---

Plan Title=Ramona Flow Control Curve
Program Version=5.01
Short Identifier=RE Flow Control Curve
Geom File=g05
Flow File=f04
Subcritical Flow
K Sum by GR= 0
Std Step Tol= 0.01
Critical Tol= 0.01
Num of Std Step Trials= 20
Max Error Tol= 0.3
Flow Tol Ratio= 0.001
Split Flow NTrial= 30
Split Flow Tol= 0.02
Split Flow Ratio= 0.02
Log Output Level= 0
Friction Slope Method= 1
Unsteady Friction Slope Method= 2
Unsteady Bridges Friction Slope Method= 1
Parabolic Critical Depth
Global Vel Dist= 0 , 0 , 0
Global Log Level= 0
CheckData=True
Encroach Param=-1 ,0,0, 0
BEGIN DESCRIPTION:
Model to develop rating curve of the Flow Control Structure from the 1974 SJR MDP.  This is taken from the 2000 WEST Model.  Elevations have been updated to NAVD 88.  Results from this model will be input into 2d Ras of Mystic Lake.
JCC  22June2016
END DESCRIPTION:
Computation Interval=1HOUR
Output Interval=1HOUR
Instantaneous Interval=1HOUR
Mapping Interval=1HOUR
Run HTab= 0
Run UNet= 0
Run Sediment= 0
Run PostProcess= 0
Run WQNet= 0
Run RASMapper= 0
UNET Theta= 1
UNET Theta Warmup= 1
UNET ZTol= 0.02
UNET ZSATol= 0.05
UNET MxIter= 20
UNET Max Iter WO Improvement= 0
UNET MaxInSteps= 0
UNET DtIC= 0
UNET DtMin= 0
UNET MaxCRTS= 20
UNET WFStab= 2
UNET SFStab= 1
UNET WFX= 1
UNET SFX= 1
UNET DSS MLevel= 4
UNET Pardiso=0
UNET DZMax Abort= 100
UNET Use Existing IB Tables=-1
UNET Froude Reduction=False
UNET Froude Limit= 1
UNET Froude Power= 10
UNET Time Slicing=0,0, 5
UNET Junction Losses=0
UNET D1 Cores= 0
UNET D2 Coriolis=0
UNET D2 Cores= 0
UNET D2 Theta= 1
UNET D2 Theta Warmup= 1
UNET D2 Z Tol= 0.01
UNET D2 Volume Tol= 0.01
UNET D2 Max Iterations= 20
UNET D2 Equation= 0
UNET D2 RampUpFraction=0.1
UNET D2 TimeSlices= 1
UNET D2 BCVolumeCheck=0
UNET D1D2 MaxIter= 0
UNET D1D2 ZTol=0.01
UNET D1D2 QTol=0.1
UNET D1D2 MinQTol=1
Write IC File= 0
Write IC File at Fixed DateTime=0
Write IC File at Sim End=0
Echo Input=False
Echo Parameters=False
Echo Output=False
Write Detailed= 0
HDF Write Warmup=0
HDF Write Time Slices=0
HDF Flush=0
HDF Face Node Velocities=0
HDF Compression= 1
HDF Chunk Size= 1
HDF Spatial Parts= 1
HDF Use Max Rows=0
HDF Fixed Rows= 1
Calibration Method= 0
Calibration Iterations= 20
Calibration Max Change=0.05
Calibration Tolerance=0.2
Calibration Maximum=1.5
Calibration Minimum=0.5
Calibration Optimization Method= 1
WQ AD Non Conservative
WQ ULTIMATE=-1
WQ Max Comp Step=1HOUR
WQ Output Interval=15MIN
WQ Output Selected Increments= 0
WQ Output face flow=0
WQ Output face velocity=0
WQ Output face area=0
WQ Output face dispersion=0
WQ Output cell volume=0
WQ Output cell surface area=0
WQ Output cell continuity=0
WQ Output cumulative cell continuity=0
WQ Output face conc=0
WQ Output face dconc_dx=0
WQ Output face courant=0
WQ Output face peclet=0
WQ Output face adv mass=0
WQ Output face disp mass=0
WQ Output cell mass=0
WQ Output cell source sink temp=0
WQ Output nsm pathways=0
WQ Output nsm derived pathways=0
WQ Output MaxMinRange=-1
WQ Daily Max Min Mean=-1
WQ Daily Range=0
WQ Daily Time=0
WQ Create Restart=0
WQ Fixed Restart=0
WQ System Summary=0
WQ Write To DSS=0
WQ Use Fixed Temperature=0
Sorting and Armoring Iterations= 10
XS Update Threshold= 0.02
Bed Roughness Predictor= 0
Hydraulics Update Threshold= 0.02
Energy Slope Method= 1
Volume Change Method= 1
Sediment Retention Method= 0
XS Weighting Method= 0
Number of US Weighted Cross Sections= 1
Number of DS Weighted Cross Sections= 1
Upstream XS Weight=0
Main XS Weight=1
Downstream XS Weight=0
Number of DS XS's Weighted with US Boundary= 1
Upstream Boundary Weight= 1
Weight of XSs Associated with US Boundary= 0
Number of US XS's Weighted with DS Boundary= 1
Downstream Boundary Weight= 0.5
Weight of XSs Associated with DS Boundary= 0.5
Percentile Method= 0
Sediment Output Level= 4
Mass or Volume Output= 0
Output Increment Type= 1
Profile and TS Output Increment= 1
XS Output Flag= 0
XS Output Increment= 10
Write Gradation File= 0
Read Gradation Hotstart= 0
Write HDF5 File= 1
Write DSS Sediment File= 0
SV Curve= 0
Specific Gage Flag= 0

--- RamonaFlowControl.f04 (steady flow) ---

Flow Title=Flow Series
Program Version=5.01
Number of Profiles= 14
Profile Names=PF 1,PF 2,PF 3,PF 4,PF 5,PF 6,PF 7,PF 8,PF 9,PF 10,PF 11,PF 12,PF 13,PF 14
River Rch & RM=San Jacinto,4               ,117440.
     250     500    1000    1500    2000    2500    3000    3500    4000    4500
    5000    5500    6000    6500
Boundary for River Rch & Prof#=San Jacinto,4               , 1
Up Type= 0
Dn Type= 2
Boundary for River Rch & Prof#=San Jacinto,4               , 2
Up Type= 0
Dn Type= 2
Boundary for River Rch & Prof#=San Jacinto,4               , 3
Up Type= 0
Dn Type= 2
Boundary for River Rch & Prof#=San Jacinto,4               , 4
Up Type= 0
Dn Type= 2
Boundary for River Rch & Prof#=San Jacinto,4               , 5
Up Type= 0
Dn Type= 2
Boundary for River Rch & Prof#=San Jacinto,4               , 6
Up Type= 0
Dn Type= 2
Boundary for River Rch & Prof#=San Jacinto,4               , 7
Up Type= 0
Dn Type= 2
Boundary for River Rch & Prof#=San Jacinto,4               , 8
Up Type= 0
Dn Type= 2
Boundary for River Rch & Prof#=San Jacinto,4               , 9
Up Type= 0
Dn Type= 2
Boundary for River Rch & Prof#=San Jacinto,4               , 10
Up Type= 0
Dn Type= 2
Boundary for River Rch & Prof#=San Jacinto,4               , 11
Up Type= 0
Dn Type= 2
Boundary for River Rch & Prof#=San Jacinto,4               , 12
Up Type= 0
Dn Type= 2
Boundary for River Rch & Prof#=San Jacinto,4               , 13
Up Type= 0
Dn Type= 2
Boundary for River Rch & Prof#=San Jacinto,4               , 14
Up Type= 0
Dn Type= 2
DSS Import GetInterval= 0
DSS Import GetPeak= 0
DSS Import FillOption= 0

--- RamonaFlowControl.g05 (geometry) ---

Geom Title=RE Flow Control Structure
Program Version=5.01
BEGIN GEOM DESCRIPTION:
This models the Flow Clontrol Structure at Ramona Expressway.  This was from the WEST model.  It was vertically adjusted 2.56 feet to be on NAVD 88.  This models the 7 cell 5'h x 10' Wide Flow Control Structure proposed in the 1974 Master Plan
JCC 22June2016
END GEOM DESCRIPTION:

River Reach=San Jacinto     ,4
Reach XY= 2
        0.465015       0.6505214      -0.0016522       0.1713422

Type RM Length L Ch R = 1 ,117440. ,1950,2005,1950
BEGIN DESCRIPTION:
WEST xsec 7500, beginning reach 4 after reach 2 & 3 rejoin.
END DESCRIPTION:
#Sta/Elev= 19
       0 1462.56     340 1458.56     850 1454.56    1440 1450.56    2020 1446.56
    2480 1442.56    2990 1438.56    3310 1434.56    4010 1430.56    4300 1426.56
    6660 1422.56    6695 1422.06    6730 1422.56    8150 1422.56    8820 1422.56
    9860 1422.56   11100 1426.56   11220 1430.56   11650 1462.56
#Mann= 3 , 0 , 0
       0    .035       0    6660     .04       0    6730    .035       0
Bank Sta=6660,6730
XS Rating Curve= 0 ,0
Exp/Cntr=0.3,0.1

Type RM Length L Ch R = 1 ,115435. ,1800,1530,1580
BEGIN DESCRIPTION:
WEST xsec 7400
END DESCRIPTION:
#Sta/Elev= 28
       0 1462.56     360 1458.56     610 1454.56    1030 1450.56    1280 1446.56
    1360 1442.56    1700 1438.56    2100 1434.56    2430 1430.56    2770 1426.56
    5250 1422.56    5285 1422.06    5320 1422.56    5330 1426.56    5380 1426.56
    5390 1423.06    6150 1422.56    6230 1422.56    6360 1422.56    6450 1422.56
    6750 1420.56    7370 1421.56    8330 1422.56    8520 1426.56    8600 1430.56
    8720 1434.56    8800 1438.56    9200 1462.56
#Mann= 3 , 0 , 0
       0    .035       0    5250     .04       0    5320    .035       0
#XS Ineff= 2 , 0
       0    2550                       0
Permanent Ineff=
       F       F
Bank Sta=5250,5320
XS Rating Curve= 0 ,0
Exp/Cntr=0.3,0.1

Type RM Length L Ch R = 1 ,113905. ,1070,1205,1270
BEGIN DESCRIPTION:
WEST xsec 7300
END DESCRIPTION:
#Sta/Elev= 23
       0 1446.56     130 1442.56     490 1438.56     700 1434.56    1100 1430.56
    1700 1426.56    2100 1422.56    3510 1422.56    3530 1418.56    3560 1418.56
    3570 1422.56    3580 1420.56    4030 1420.56    4080 1418.56    4110 1418.56
    4120 1420.56    5610 1422.56    6320 1426.56    6420 1430.56    6510 1434.56
    6590 1438.56    6650 1442.56    6710 1446.56
#Mann= 3 , 0 , 0
       0    .035       0    3510     .04       0    3570    .035       0
#XS Ineff= 2 , 0
       0    1700                       0
Permanent Ineff=
       F       F
Bank Sta=3510,3570
XS Rating Curve= 0 ,0
Exp/Cntr=0.3,0.1

Type RM Length L Ch R = 1 ,112700. ,810,970,1000
BEGIN DESCRIPTION:
WEST xsec 7200
END DESCRIPTION:
#Sta/Elev= 14
       0 1438.56     310 1434.56     640 1430.56    1160 1426.56    1480 1422.56
    2850 1422.56    2910 1418.56    2950 1418.56    2980 1422.56    4680 1422.56
    5150 1426.56    5300 1430.56    5380 1434.56    5450 1438.56
#Mann= 3 , 0 , 0
       0    .035       0    2850    .035       0    2980    .035       0
#XS Ineff= 2 , 0
       0    1650 1435.61    4450       0 1438.86
Permanent Ineff=
       F       F
Bank Sta=2850,2980
XS Rating Curve= 0 ,0
Exp/Cntr=0.3,0.1

Type RM Length L Ch R = 1 ,111730. ,330,330,330
BEGIN DESCRIPTION:
WEST sta/elev data at RCFCD xsec 71 location
END DESCRIPTION:
#Sta/Elev= 12
       0 1434.56     230 1430.56     920 1426.56    1370 1422.56    2690 1422.56
    2700 1418.56    2730 1418.56    2750 1422.56    3460 1422.56    4490 1426.56
    4590 1430.56    4720 1434.56
#Mann= 3 , 0 , 0
       0    .035       0    2690    .035       0    2750    .035       0
#XS Ineff= 2 , 0
       0    2000 1435.61    3250       0 1438.86
Permanent Ineff=
       F       F
Bank Sta=2690,2750
XS Rating Curve= 0 ,0
Exp/Cntr=0.3,0.1

Type RM Length L Ch R = 1 ,111400. ,225,225,225
BEGIN DESCRIPTION:
This is xsec 7000 (RCFCD data  from xsec 200100 to 207000) modified to U/S face of Ramona Expressway Bridge and adjusted to fit bridge approach.  The updated data comes from RCFC&WCD San Jancinto River map, portion of section T4SR2W,Sheet 5 of 13.  Greater topo detail was avialable from this map for the approach roads to the bridge from both directions. GR data was taken on the center line of the road from the edge of bridge crossing to the outer banks.
END DESCRIPTION:
#Sta/Elev= 30
       0 1436.16   517.1 1430.96   899.1 1428.66  1284.7 1425.86  1367.8 1424.66
  1836.4 1422.56  2052.3 1422.36  2305.1 1422.36  2595.2 1422.76    2598 1422.86
    2628 1426.46  2656.6 1427.06  2685.9 1421.36  2715.2 1419.96  2771.9 1419.76
  2773.8 1419.76  2803.1 1423.06  2819.9 1427.66  2832.4 1430.06  2861.7 1423.26
  2867.9 1423.06    2891 1422.86  2923.2 1422.76  3242.4 1422.96  3587.4 1422.36
  3711.1 1421.76  4179.7 1422.36    4355 1424.36  4684.4 1429.16  4988.8 1444.16
#Mann= 3 , 0 , 0
       0    .035       0  2656.6    .035       0  2832.4    .035       0
#XS Ineff= 2 , 0
       0    2405 1435.61    3095       0 1438.86
Permanent Ineff=
       F       F
Bank Sta=2656.6,2832.4
XS Rating Curve= 0 ,0
Exp/Cntr=0.3,0.1

Type RM Length L Ch R = 1 ,111175. ,50,50,50
BEGIN DESCRIPTION:
This is xsec 7000 (RCFCD data  from xsec 200100 to 207000) modified to U/S face of Ramona Expressway Bridge and adjusted to fit bridge approach.  The updated data comes from RCFC&WCD San Jancinto River map, portion of section T4SR2W,Sheet 5 of 13.  Greater topo detail was avialable from this map for the approach roads to the bridge from both directions. GR data was taken on the center line of the road from the edge of bridge crossing to the outer banks.
END DESCRIPTION:
#Sta/Elev= 24
       0 1436.16   430.4 1431.76   517.1 1430.96   899.1 1428.66  1284.7 1425.86
  1367.8 1424.66  1836.4 1422.56  2052.3 1422.36  2305.1 1422.36    2530 1422.56
  2555.5 1430.56  2605.5 1430.56  2618.1 1419.56  2839.7 1419.56  2856.1 1430.56
  2906.1 1430.56    2927 1422.56  3242.4 1422.96  3587.4 1422.36  3711.1 1421.76
  4179.7 1422.36    4355 1424.36  4684.4 1429.16  4988.8 1444.16
#Mann= 3 , 0 , 0
       0    .035       0  2605.5    .035       0  2856.1    .035       0
#XS Ineff= 2 , 0
       0  2605.5 1435.61  2856.1       0 1438.86
Permanent Ineff=
       F       F
Bank Sta=2605.5,2856.1
XS Rating Curve= 0 ,0
Exp/Cntr=0.3,0.1

Type RM Length L Ch R = 3 ,111150. ,,,
BEGIN DESCRIPTION:
Existing Ramona Expressway Bridge
Bridge piers were modeled twice the size to accomodate the piers that are behind the front piers.  This was done to represent the 10 degree skew.  The levees were modeled to what the plans and field notes show.  The overlaying area were taken from the topo maps.
END DESCRIPTION:
Bridge Culvert-0,0,-1,-1, 0
Deck Dist Width WeirC Skew NumUp NumDn MinLoCord MaxHiCord MaxSubmerge Is_Ogee
10,30,2.6,0, 41, 41, , , 0.95, 0, 1,1,,
       0     400     800    1685    2355  2538.7  2538.7    2600    2600 2605.25
 2605.25  2605.5  2605.5    2705    2770  2782.4    2850  2852.3  2852.3  2856.7
 2861.25 2861.25  2862.6  2862.6  2927.7  2927.7    2940    2970    3000    3015
    3315    4015    4400    4405    4425    4430    4555    4750    5100    5160
    5220
 1438.56 1434.56 1430.56 1429.56 1430.56 1430.56 1433.31 1433.31 1433.31 1433.31
 1433.31 1433.31 1433.31 1433.31 1433.31 1433.31 1433.31 1433.31 1433.31 1433.31
 1433.31 1433.31 1433.31 1433.31 1433.31 1430.56 1430.56 1430.56 1430.56 1430.56
 1430.56 1429.56 1428.56 1428.56 1428.56 1428.56 1429.56 1430.56 1434.56 1438.56
 1442.56
                                                                                
                 1429.26 1429.26 1429.26 1429.26 1429.26 1429.26
                                                                                
                                                                                
        
       0     400     800    1685    2355  2538.7  2538.7    2600    2600 2605.25
 2605.25  2605.5  2605.5    2705    2770  2782.4    2850  2852.3  2852.3  2856.7
 2861.25 2861.25  2862.6  2862.6  2927.7  2927.7    2940    2970    3000    3015
    3315    4015    4400    4405    4425    4430    4555    4750    5100    5160
    5220
 1438.56 1434.56 1430.56 1429.56 1430.56 1430.56 1433.31 1433.31 1433.31 1433.31
 1433.31 1433.31 1433.31 1433.31 1433.31 1433.31 1433.31 1433.31 1433.31 1433.31
 1433.31 1433.31 1433.31 1433.31 1433.31 1430.56 1430.56 1430.56 1430.56 1430.56
 1430.56 1429.56 1428.56 1428.56 1428.56 1428.56 1429.56 1430.56 1434.56 1438.56
 1442.56
                                                                                
                 1429.26 1429.26 1429.26 1429.26 1429.26 1429.26
                                                                                
                                                                                
        
Pier Skew, UpSta & Num, DnSta & Num=  ,2623.65, 2 ,2623.65, 2 , 0 , 0 , 0 ,,
     2.6     2.6
 1387.56 1430.56
     2.6     2.6
 1387.56 1430.56
Pier Skew, UpSta & Num, DnSta & Num=  ,2645.31, 2 ,2645.31, 2 , 0 , 0 , 0 ,,
     2.6     2.6
 1387.56 1430.56
     2.6     2.6
 1387.56 1430.56
Pier Skew, UpSta & Num, DnSta & Num=  ,2666.97, 2 ,2666.97, 2 , 0 , 0 , 0 ,,
     2.6     2.6
 1387.56 1430.56
     2.6     2.6
 1387.56 1430.56
Pier Skew, UpSta & Num, DnSta & Num=  ,2688.63, 2 ,2688.63, 2 , 0 , 0 , 0 ,,
     2.6     2.6
 1387.56 1430.56
     2.6     2.6
 1387.56 1430.56
Pier Skew, UpSta & Num, DnSta & Num=  ,2710.29, 2 ,2710.29, 2 , 0 , 0 , 0 ,,
     2.6     2.6
 1387.56 1430.56
     2.6     2.6
 1387.56 1430.56
Pier Skew, UpSta & Num, DnSta & Num=  ,2731.95, 2 ,2731.95, 2 , 0 , 0 , 0 ,,
     2.6     2.6
 1387.56 1430.56
     2.6     2.6
 1387.56 1430.56
Pier Skew, UpSta & Num, DnSta & Num=  ,2753.61, 2 ,2753.61, 2 , 0 , 0 , 0 ,,
     2.6     2.6
 1387.56 1430.56
     2.6     2.6
 1387.56 1430.56
Pier Skew, UpSta & Num, DnSta & Num=  ,2775.27, 2 ,2775.27, 2 , 0 , 0 , 0 ,,
     2.6     2.6
 1387.56 1430.56
     2.6     2.6
 1387.56 1430.56
Pier Skew, UpSta & Num, DnSta & Num=  ,2796.93, 2 ,2796.93, 2 , 0 , 0 , 0 ,,
     2.6     2.6
 1387.56 1430.56
     2.6     2.6
 1387.56 1430.56
Pier Skew, UpSta & Num, DnSta & Num=  ,2818.59, 2 ,2818.59, 2 , 0 , 0 , 0 ,,
     2.6     2.6
 1387.56 1430.56
     2.6     2.6
 1387.56 1430.56
Pier Skew, UpSta & Num, DnSta & Num=  ,2840.25, 2 ,2840.25, 2 , 0 , 0 , 0 ,,
     2.6     2.6
 1387.56 1430.56
     2.6     2.6
 1387.56 1430.56
BR Coef=-1 , 1 , 0 ,0.9, 0 ,,,0.8,-1,1.2,0,
WSPro=,,,, 1 ,,,, 0 ,,,, 0 ,,,,-1 ,-1 ,-1 , 0 , 0 , 0 , 0 , 0
BC Design=,, 0 ,, 0 ,,,,,,
BC HTab HWMax=1444.16
BC Use User HTab Curves=0
BC User HTab FreeFlow(D)= 0

Type RM Length L Ch R = 1 ,111125. ,15,15,15
BEGIN DESCRIPTION:
This is a copy of xsec 6990 (RCFCD data  from xsec 200100 to 207000) copied to D/S face of Ramona Expressway Bridge
(this section was copied from 206800)
END DESCRIPTION:
#Sta/Elev= 24
       0 1436.16   430.4 1431.76   517.1 1430.96   899.1 1428.66  1284.7 1425.86
  1367.8 1424.66  1836.4 1422.56  2052.3 1422.36  2305.1 1422.36    2530 1422.56
  2555.5 1430.56  2605.5 1430.56  2617.7 1419.56  2839.3 1419.56  2856.1 1430.56
  2906.1 1430.56    2927 1422.56  3242.4 1422.96  3587.4 1422.36  3711.1 1421.76
  4179.7 1422.36    4355 1424.36  4684.4 1429.16  4988.8 1444.16
#Mann= 3 , 0 , 0
       0     .03       0  2605.5    .035       0  2856.1     .03       0
#XS Ineff= 2 , 0
       0 2598.43 1435.61 2854.33       0 1438.86
Permanent Ineff=
       F       F
Bank Sta=2605.5,2856.1
XS Rating Curve= 0 ,0
Exp/Cntr=0.3,0.1

Type RM Length L Ch R = 1 ,111110  ,138,138,138
BEGIN DESCRIPTION:
20 feet u/s of culvert face
END DESCRIPTION:
#Sta/Elev= 29
       0 1436.16   430.4 1431.76   517.1 1430.96   899.1 1428.66  1284.7 1425.86
  1367.8 1424.66  1836.4 1422.56    2530 1422.56    2615 1423.56    2622 1424.56
    2630 1426.56    2637 1427.16    2646 1426.56    2657 1423.56    2662 1422.56
    2670 1421.56  2670.8 1418.58  2786.2 1418.58  2786.5 1421.56    2793 1422.56
    2802 1424.56    2808 1425.56    2821 1430.56    2849 1430.56    2865 1423.56
    2870 1422.56    4355 1424.36  4684.4 1429.16  4988.8 1444.16
#Mann= 3 , 0 , 0
       0     .03       0    2637    .035       0    2821     .03       0
#XS Ineff= 2 , 0
       0  2670.8 1435.61  2786.2       0 1438.86
Permanent Ineff=
       F       F
Bank Sta=2637,2821
XS Rating Curve= 0 ,0
Exp/Cntr=0.3,0.1

Type RM Length L Ch R = 2 ,111041  ,,,
BEGIN DESCRIPTION:
Proposed 7 - 10 X 5 culverts for eastbound Ramona
END DESCRIPTION:
Bridge Culvert--1,0,-1,-1, 0
Deck Dist Width WeirC Skew NumUp NumDn MinLoCord MaxHiCord MaxSubmerge Is_Ogee
47,42,3,0, 10, 10, , , 0.95, 0, 4,4,,
       0  2060.5  2260.5  2360.5  2460.5  3060.5  3161.5  3261.5  4684.4  4988.8
 1436.56 1436.86 1435.86 1435.61 1435.86 1438.86 1439.11 1438.86 1438.56 1444.16
                                                                                
       0  2060.5  2260.5  2360.5  2460.5  3060.5  3161.5  3261.5  4684.4  4988.8
 1436.56 1436.86 1435.86 1435.61 1435.86 1438.86 1439.11 1438.86 1438.56 1444.16
                                                                                
Multiple Barrel Culv=2,5,10,97.73,0.011,0.5,1,8,1,1418.58,1418.56, 7,Culvert #1  , 0 ,20
 2696.49 2712.09 2707.16 2722.76 2717.83 2733.43  2728.5  2744.1 2739.17 2754.77
 2749.84 2765.44 2760.51 2776.11
Culvert Bottom n=0.011
BC Design=,, 0 ,, 0 ,,,,,,
BC HTab HWMax=1444.16
BC Use User HTab Curves=0
BC User HTab FreeFlow(D)= 0

Type RM Length L Ch R = 1 ,110972  ,62,62,62
BEGIN DESCRIPTION:
20.27 feet d/s of culvert face
END DESCRIPTION:
#Sta/Elev= 30
       0 1436.16   430.4 1431.76   517.1 1430.96   899.1 1428.66  1284.7 1425.86
  1367.8 1424.66  1836.4 1422.56  2052.3 1422.36  2305.1 1422.36  2595.2 1422.76
    2598 1422.86    2628 1426.46  2656.6 1427.06  2685.9 1421.36  2686.4 1418.56
  2801.8 1418.56  2803.1 1423.06  2819.9 1427.66  2832.4 1430.06  2861.7 1423.26
  2867.9 1423.06    2891 1422.86  2923.2 1422.76  3242.4 1422.96  3587.4 1422.36
  3711.1 1421.76  4179.7 1422.36    4355 1424.36  4684.4 1429.16  4988.8 1444.16
#Mann= 3 , 0 , 0
       0     .03       0  2656.6    .035       0  2832.4     .03       0
#XS Ineff= 2 , 0
       0  2701.6 1434.61  2786.6       0 1438.16
Permanent Ineff=
       F       F
Bank Sta=2656.6,2832.4
XS Rating Curve= 0 ,0
Exp/Cntr=0.3,0.1

Type RM Length L Ch R = 1 ,110910. ,500,500,500
BEGIN DESCRIPTION:
6800
END DESCRIPTION:
#Sta/Elev= 30
       0 1436.16   517.1 1430.96   899.1 1428.66  1284.7 1425.86  1367.8 1424.66
  1836.4 1422.56  2052.3 1422.36  2305.1 1422.36  2595.2 1422.76    2598 1422.86
    2628 1426.46  2656.6 1427.06  2685.9 1421.36  2715.2 1419.96  2771.9 1419.76
  2773.8 1419.76  2803.1 1423.06  2819.9 1427.66  2832.4 1430.06  2861.7 1423.26
  2867.9 1423.06    2891 1422.86  2923.2 1422.76  3242.4 1422.96  3587.4 1422.36
  3711.1 1421.76  4179.7 1422.36    4355 1424.36  4684.4 1429.16  4988.8 1444.16
#Mann= 3 , 0 , 0
       0     .03       0  2656.6    .035       0  2832.4     .03       0
#XS Ineff= 2 , 0
       0  2689.5 1434.56  2799.5       0 1437.56
Permanent Ineff=
       F       F
Bank Sta=2656.6,2832.4
XS Rating Curve= 0 ,0
Exp/Cntr=0.3,0.1

Type RM Length L Ch R = 1 ,110410. ,505,505,505
BEGIN DESCRIPTION:
6700
END DESCRIPTION:
#Sta/Elev= 30
       0 1431.96    49.6 1431.46     518 1428.76   776.1 1426.66   986.5 1424.56
    1455 1421.46  1544.5 1421.36  1923.4 1422.26    1982 1421.76  2011.3 1423.76
  2024.8 1423.36  2040.6 1421.96  2069.9 1420.16  2072.9 1420.36  2128.4 1418.86
  2157.7 1419.66    2187 1419.56  2216.3 1420.26  2245.6 1424.36    2265 1428.66
  2274.8 1429.26  2304.1 1422.56  2391.9 1421.86  2860.4 1421.26  3081.4 1422.06
  3328.9 1423.66  3797.3 1424.06  3849.9 1421.86  4265.8 1431.16  4300.9 1432.76
#Mann= 3 , 0 , 0
       0     .03       0  2011.3    .035       0  2274.8     .03       0
#XS Ineff= 2 , 0
       0    1910 1434.56    2440       0 1437.56
Permanent Ineff=
       F       F
Bank Sta=2011.3,2274.8
XS Rating Curve= 0 ,0
Exp/Cntr=0.3,0.1

Type RM Length L Ch R = 1 ,109905. ,505,505,505
BEGIN DESCRIPTION:
6600
END DESCRIPTION:
#Sta/Elev= 30
       0 1431.56   198.8 1430.26     667 1428.66   774.4 1427.76  1135.2 1423.86
  1543.9 1422.16  1603.4 1422.06  2024.2 1421.26  2042.4 1421.16  2071.7 1421.76
    2073 1421.96  2100.9 1422.86  2121.1 1420.06  2130.2 1419.16  2159.4 1418.86
  2169.2 1418.86  2188.7 1418.86    2218 1420.56  2247.2 1426.26  2265.4 1428.26
  2276.5 1427.36  2305.8 1421.86  2313.5 1421.66  2333.3 1421.46  2539.9 1421.26
  3008.1 1423.96    3083 1423.96  3476.3 1424.56  3944.5 1423.66  4403.4 1433.16
#Mann= 3 , 0 , 0
       0     .03       0  2100.9    .035       0  2265.4     .03       0
#XS Ineff= 2 , 0
       0    1710 1434.56    2690       0 1437.56
Permanent Ineff=
       F       F
Bank Sta=2100.9,2265.4
XS Rating Curve= 0 ,0
Exp/Cntr=0.3,0.1

Type RM Length L Ch R = 1 ,109400. ,490,490,490
BEGIN DESCRIPTION:
6500
END DESCRIPTION:
#Sta/Elev= 28
       0 1430.46   147.4 1429.26   601.8 1427.56  1084.5 1423.56  1369.8 1422.66
  1553.1 1422.26    1841 1421.26  1893.5 1421.36  1934.9 1423.06  1981.4 1420.26
  1982.9 1420.36  2010.7 1418.06  2030.9 1415.96    2040 1416.56  2078.9 1426.76
  2098.5 1429.66  2127.8 1422.06  2157.1 1421.36  2174.9 1421.56  2186.4 1421.76
  2215.7 1421.76  2230.6 1421.76  2490.2 1423.16  2958.8 1424.16  3427.4 1424.16
  3673.9 1424.46  3895.9 1425.96  4238.6 1433.36
#Mann= 3 , 0 , 0
       0     .03       0  1934.9    .035       0  2098.5     .03       0
Bank Sta=1934.9,2098.5
XS Rating Curve= 0 ,0
Exp/Cntr=0.3,0.1

Type RM Length L Ch R = 1 ,108910. ,505,505,505
BEGIN DESCRIPTION:
6400
WEST:  Measured from zero back 120 feet to obtain elevation 1428.  Then added 120 constant to all stationing in order to remove of the negative 120 feet measurement. (RCFCD photo maps)
END DESCRIPTION:
#Sta/Elev= 30
       0 1430.56     120 1429.46   506.7 1428.76   788.4 1427.36   974.3 1426.16
  2061.3 1420.86  2140.3 1420.66  2172.4 1420.66  2188.6 1422.46  2201.6 1422.96
  2230.9 1420.46  2236.9 1420.66  2260.1 1419.06  2285.2 1416.26  2289.3 1416.46
  2318.5 1423.26  2333.4 1426.26  2347.7 1428.76    2377 1424.36  2381.7 1423.36
  2406.2 1421.76    2430 1421.66  2435.4 1422.06  2844.5 1423.56    3106 1423.46
  3312.1 1423.16  3779.6 1423.26  3878.5 1423.86  4247.2 1428.36  4328.7 1431.16
#Mann= 3 , 0 , 0
       0     .03       0  2201.6    .035       0  2347.7     .03       0
#XS Ineff= 2 , 0
       0                    3701       0 1437.56
Permanent Ineff=
       F       F
Bank Sta=2201.6,2347.7
XS Rating Curve= 0 ,0
Exp/Cntr=0.3,0.1

Type RM Length L Ch R = 1 ,108405. ,510,510,510
BEGIN DESCRIPTION:
6300
END DESCRIPTION:
#Sta/Elev= 28
       0 1430.86     126 1424.06   594.1 1425.76  1062.2 1424.46  1530.3 1422.26
    1532 1423.56  1998.4 1421.56  2064.9 1421.46  2086.2 1421.36  2144.7 1421.66
  2173.9 1423.36  2203.2 1421.16  2205.8 1420.86  2232.5 1418.76  2253.9 1418.46
  2261.7 1418.56    2291 1419.66    2302 1420.56  2349.5 1428.86  2378.7 1422.16
  2398.3 1421.86  2466.5 1421.86  2934.6 1422.76  3072.1 1422.36  3402.7 1421.96
  3842.2 1422.66  3870.8 1422.76  4306.2 1437.66
#Mann= 3 , 0 , 0
       0     .03       0  2173.9    .035       0  2349.5     .03       0
#XS Ineff= 2 , 0
       0                    3560       0 1437.56
Permanent Ineff=
       F       F
Bank Sta=2173.9,2349.5
XS Rating Curve= 0 ,0
Exp/Cntr=0.3,0.1

Type RM Length L Ch R = 1 ,107895. ,490,490,490
BEGIN DESCRIPTION:
6200
WEST:  Measured back from zero 350 feet to obtain 1428 ft. elevation.  Added 350 constant to all stationing in order to remove -350 feet measurement. (RCFCD photo maps)
END DESCRIPTION:
#Sta/Elev= 29
       0 1430.56     350 1428.56   616.8 1422.56  1085.6 1424.56  1554.4 1425.06
  1883.7 1424.76  2023.3 1421.86  2492.1 1423.56  2561.3 1420.96  2579.6 1421.06
  2594.2 1421.66  2608.9 1422.76  2638.2 1423.66  2667.5 1418.96  2696.8 1416.96
  2726.1 1417.86    2738 1419.26  2755.4 1426.36  2784.7 1426.46  2785.9 1426.16
    2814 1422.46  2833.8 1421.86  2843.3 1421.76  2960.9 1421.96  3429.8 1421.96
    3898 1421.56  4184.1 1422.26  4367.5 1426.06  4510.7 1430.76
#Mann= 3 , 0 , 0
       0     .03       0  2638.2    .035       0  2784.7     .03       0
#XS Ineff= 2 , 0
       0                    3190       0 1437.56
Permanent Ineff=
       F       F
Bank Sta=2638.2,2784.7
XS Rating Curve= 0 ,0
Exp/Cntr=0.3,0.1

Type RM Length L Ch R = 1 ,107405. ,475,475,475
BEGIN DESCRIPTION:
6100
WEST: Measured back from zero 550 feet to obtain 1428 ft. elevation.  Added 550 feet constant to start at 0 . (RCFCD photo maps)
END DESCRIPTION:
#Sta/Elev= 30
       0 1430.56     550 1428.26   918.3 1422.56  1017.9 1422.46  1485.7 1424.16
  1689.4 1423.46  1953.6 1421.76  2421.5 1420.86  2804.7 1421.16  2833.9 1421.66
  2874.6 1423.66  2892.4 1422.86  2921.6 1417.96  2950.9 1417.36    2971 1418.26
  2980.1 1419.06  3009.4 1425.26  3019.2 1426.46  3038.6 1426.16  3067.8 1422.36
  3099.2 1422.16  3357.2 1422.36    3825 1420.36  3991.4 1422.56  4002.8 1421.06
  4191.4 1422.56  4291.4 1426.56  4292.9 1425.86  4431.4 1430.56  4503.3 1434.46
#Mann= 3 , 0 , 0
       0     .03       0  2874.6    .035       0  3019.2     .03       0
#XS Ineff= 2 , 0
       0     860 1434.56    3940       0 1437.56
Permanent Ineff=
       F       F
Bank Sta=2874.6,3019.2
XS Rating Curve= 0 ,0
Exp/Cntr=0.3,0.1

Type RM Length L Ch R = 1 ,106930. ,505,505,505
BEGIN DESCRIPTION:
6000
WEST:  Measured back from zero 350 feet to obtain 1428 ft elevation.  Added 270 feet to remove negative number. (RCFCD photo maps)
END DESCRIPTION:
#Sta/Elev= 29
       0 1430.56     270 1427.46   502.4 1424.56     737 1423.76  1277.7 1423.06
  1670.8 1421.86    2053 1423.76  2137.8 1423.96  2568.4 1421.26  2580.5 1421.56
  2609.7 1421.76  2622.9 1422.26  2638.9 1422.76  2668.1 1421.76  2697.3 1419.56
  2719.8 1418.66  2726.5 1418.56  2755.7 1419.36  2768.3 1421.36  2784.8 1424.96
    2814 1427.06  2843.2 1424.36  2865.2 1424.36  2872.4 1424.46  2899.7 1424.36
  3071.7 1422.16  3603.5 1421.76  4005.6 1427.86  4158.8 1432.86
#Mann= 3 , 0 , 0
       0     .03       0  2638.9    .035       0    2814     .03       0
#XS Ineff= 2 , 0
       0     710 1434.56               0
Permanent Ineff=
       F       F
Bank Sta=2638.9,2814
XS Rating Curve= 0 ,0
Exp/Cntr=0.3,0.1

Type RM Length L Ch R = 1 ,106425. ,505,505,505
BEGIN DESCRIPTION:
5900
WEST:  Measured back from zero 350 feet to obtain 1428 ft elevation.  Added 350 feet constant to all stations to correct zero. (RCFCD photo maps)
END DESCRIPTION:
#Sta/Elev= 30
       0 1430.56     350 1427.26   816.7 1423.96   958.1 1423.66  1283.5 1423.16
  1750.2 1422.86  2216.9 1423.46  2510.7 1423.06  2683.7 1422.46  2733.5 1421.56
  2771.5 1421.26  2778.7 1421.36  2807.9 1424.76    2820 1423.46  2837.1 1420.56
  2866.2 1416.86  2895.4 1417.76  2917.1 1420.46  2924.6 1421.76  2953.7 1429.76
  2965.6 1428.66  2982.9 1424.76  3012.1 1421.66  3041.2 1422.16  3061.8 1422.06
  3150.4 1423.56    3287 1423.46  4083.9 1420.66  4550.6 1424.96    4767 1432.26
#Mann= 3 , 0 , 0
       0     .03       0  2807.9    .035       0  2953.7     .03       0
#XS Ineff= 2 , 0
       0     560 1434.56               0
Permanent Ineff=
       F       F
Bank Sta=2807.9,2953.7
XS Rating Curve= 0 ,0
Exp/Cntr=0.3,0.1

Type RM Length L Ch R = 1 ,105920. ,515,515,515
BEGIN DESCRIPTION:
5800
WEST:  Measured 600 feet back from zero to obtain 1428 ft elevation.  Added 600 constant to all stations (RCFCD photo maps)
END DESCRIPTION:
#Sta/Elev= 30
       0 1430.56   665.5 1426.06   995.7 1423.96  1440.3 1422.76  1893.8 1422.96
  2215.2 1422.66  2360.8 1422.66  2711.2 1420.76  2740.3 1420.86  2747.9 1421.26
  2769.5 1423.16  2796.3 1419.86  2798.7 1419.36  2844.7 1416.96  2857.1 1416.66
  2886.3 1420.06  2893.2 1422.26  2915.5 1428.86  2941.6 1423.26  2944.7 1422.36
  2973.9 1420.86  2999.3 1420.96  3294.9 1422.86  3764.8 1423.76    4229 1421.86
  4696.1 1422.36  5163.1 1425.16  5314.5 1426.46  5630.2 1433.86  5688.3 1436.06
#Mann= 3 , 0 , 0
       0     .03       0  2769.5    .035       0  2915.5     .03       0
Bank Sta=2769.5,2915.5
XS Rating Curve= 0 ,0
Exp/Cntr=0.3,0.1

Type RM Length L Ch R = 1 ,105405. ,495,495,495
BEGIN DESCRIPTION:
5700
WEST:  Measured back from zero 700 feet to obtain 1428 elevation.  Added 700 constant to all stations (RCFCD photo maps)
END DESCRIPTION:
#Sta/Elev= 30
       0 1430.56     700 1427.46   784.4 1425.86   879.4 1425.36  1252.5 1423.96
  1649.3 1423.16  2419.2 1422.16    2891 1420.66  2900.4 1420.86  2920.2 1422.46
  2948.5 1422.16  2949.5 1421.96  2978.8 1419.76  2996.6 1418.06    3008 1415.96
  3037.3 1418.46  3044.7 1420.06  3066.6 1425.26  3092.9 1425.16  3125.1 1420.66
    3141 1420.76  3166.6 1420.36  3593.2 1422.36    3959 1423.56  4061.4 1423.76
  4529.5 1422.46  4728.9 1422.16  4997.6 1422.26  5465.8 1424.26  5756.8 1431.46
#Mann= 3 , 0 , 0
       0     .03       0  2920.2    .035       0  3066.6     .03       0
#XS Ineff= 2 , 0
       0     900 1430.56               0
Permanent Ineff=
       F       F
Bank Sta=2920.2,3066.6
XS Rating Curve= 0 ,0
Exp/Cntr=0.3,0.1

Type RM Length L Ch R = 1 ,104910. ,505,505,505
BEGIN DESCRIPTION:
5600
WEST:  Measured back from zero 470 feet to obtain 1428 ft elevation.  Added a 470 constant to all stations. (RCFCD photo maps)
END DESCRIPTION:
#Sta/Elev= 30
       0 1430.56   739.2 1425.26    1207 1423.26  1488.8 1422.86  2142.4 1421.66
  2260.5 1421.66  2610.1 1421.96    2657 1420.96  2697.8 1420.46  2727.1 1421.26
  2742.9 1422.36  2756.3 1422.46  2791.1 1420.86  2814.8 1418.36  2839.4 1417.46
    2844 1417.86  2873.3 1425.16  2887.6 1426.66  2902.5 1426.16  2931.7 1420.76
  2935.9 1420.66  3077.9 1421.26  3545.6 1422.16  3804.1 1421.46    4481 1421.56
  4575.8 1421.66  4948.8 1420.96  5347.6 1426.46  5416.5 1428.06  5649.5 1433.06
#Mann= 3 , 0 , 0
       0     .03       0  2756.3    .035       0  2887.6     .03       0
#XS Ineff= 2 , 0
       0     900 1430.56               0
Permanent Ineff=
       F       F
Bank Sta=2756.3,2887.6
XS Rating Curve= 0 ,0
Exp/Cntr=0.3,0.1

Type RM Length L Ch R = 1 ,104405. ,490,490,490
BEGIN DESCRIPTION:
5500
END DESCRIPTION:
#Sta/Elev= 30
       0 1432.46   260.9 1429.66   727.6 1427.86  1194.2 1425.36  1808.3 1422.76
  2127.6 1422.16  2594.3 1421.76  2939.8 1420.86  3021.6 1420.06  3031.8 1420.26
    3061 1421.66  3070.1 1420.86  3090.1 1418.46  3118.6 1417.46  3148.5 1416.86
  3167.2 1420.76  3177.6 1423.36  3206.8 1426.96    3236 1420.56  3264.2 1420.06
  3276.9 1420.06  3361.3 1419.16  3527.6 1420.36    4137 1422.26    4461 1421.66
  4927.7 1419.16  5394.4 1421.46  5690.8 1425.06  5861.1 1428.46    5939 1430.96
#Mann= 3 , 0 , 0
       0     .03       0    3061    .035       0  3206.8     .03       0
#XS Ineff= 2 , 0
       0    1500 1430.56               0
Permanent Ineff=
       F       F
Bank Sta=3061,3206.8
XS Rating Curve= 0 ,0
Exp/Cntr=0.3,0.1

Type RM Length L Ch R = 1 ,103915. ,505,505,505
BEGIN DESCRIPTION:
5400
END DESCRIPTION:
#Sta/Elev= 30
       0 1432.76   313.1 1429.96   407.7 1429.46  1086.3 1427.06  1342.5 1425.86
  1809.9 1423.36  2277.3 1421.86  2632.9 1421.16  2744.7 1421.16  3017.8 1420.86
  3036.9 1421.06  3066.1 1422.06  3095.3 1419.16  3116.2 1417.46  3124.5 1417.06
  3153.7 1416.36  3164.5 1417.56  3182.9 1421.16  3212.2 1429.16  3241.4 1421.66
  3261.2 1420.16  3270.6 1419.86  3406.1 1420.36  3679.5 1420.26  4146.9 1420.66
  4614.3 1420.36  5081.7 1421.06  5549.1 1425.16  5725.8 1428.16  5949.1 1433.36
#Mann= 3 , 0 , 0
       0     .03       0  3066.1    .035       0  3212.2     .03       0
#XS Ineff= 2 , 0
       0    1500 1430.56               0
Permanent Ineff=
       F       F
Bank Sta=3066.1,3212.2
XS Rating Curve= 0 ,0
Exp/Cntr=0.3,0.1

Type RM Length L Ch R = 1 ,103410. ,495,495,495
BEGIN DESCRIPTION:
5300
END DESCRIPTION:
#Sta/Elev= 30
       0 1427.86   247.6 1425.96    1114 1422.46  1649.3 1421.76  2116.5 1420.76
  2214.1 1420.16  2262.5 1420.46    2275 1420.66  2291.7 1421.36  2323.4 1418.46
  2350.1 1417.26  2371.8 1416.66  2379.3 1416.26  2408.5 1418.86  2420.1 1421.86
  2437.7 1426.16  2466.9 1422.66  2468.5 1422.36  2496.1 1419.76  2583.7 1419.16
    2662 1419.86  3050.9 1420.56    3436 1421.46  3518.2 1421.46  3985.4 1420.36
    4210 1420.96  4452.6 1422.66  4919.9 1431.56    4984 1433.16  5138.9 1436.46
#Mann= 3 , 0 , 0
       0     .03       0  2291.7    .035       0  2437.7     .03       0
#XS Ineff= 2 , 0
       0     700 1430.56               0
Permanent Ineff=
       F       F
Bank Sta=2291.7,2437.7
XS Rating Curve= 0 ,0
Exp/Cntr=0.3,0.1

Type RM Length L Ch R = 1 ,102915. ,525,525,525
BEGIN DESCRIPTION:
5200
END DESCRIPTION:
#Sta/Elev= 30
       0 1429.26   407.4 1424.46   423.3 1424.46  1185.3 1421.96  1356.1 1421.66
  1822.4 1421.06  1963.1 1421.06  2210.9 1420.06  2288.9 1420.16  2303.4 1420.36
    2318 1420.76  2347.2 1420.76  2376.3 1417.06  2400.7 1417.36  2405.5 1417.26
  2434.6 1415.26  2449.3 1417.26  2463.8 1420.66  2492.9 1424.76  2497.9 1423.66
  2522.1 1419.56  2539.9 1419.46    2741 1419.76  2755.2 1420.36    3688 1419.76
  4154.4 1419.86  4296.7 1420.26  4620.8 1425.86  5074.5 1433.86  5183.7 1435.96
#Mann= 3 , 0 , 0
       0     .03       0  2347.2    .035       0  2492.9     .03       0
#XS Ineff= 2 , 0
       0     500 1430.56               0
Permanent Ineff=
       F       F
Bank Sta=2347.2,2492.9
XS Rating Curve= 0 ,0
Exp/Cntr=0.3,0.1

Type RM Length L Ch R = 1 ,102390. ,500,500,500
BEGIN DESCRIPTION:
5100
END DESCRIPTION:
#Sta/Elev= 30
       0 1431.26    26.1 1430.86   342.5 1427.66   491.9 1426.46   957.8 1421.96
  1122.8 1421.16  1423.6 1420.56  1889.5 1420.46  1903.2 1420.16  2144.2 1420.46
  2195.9 1420.26  2209.8 1419.96  2238.9 1420.16    2268 1421.26  2297.1 1417.46
  2326.3 1416.16  2342.3 1415.26  2355.4 1416.26  2384.5 1421.26    2391 1422.86
  2413.6 1424.96  2439.8 1419.86  2442.7 1419.66    2461 1419.46    3287 1419.66
  3752.9 1419.56  4244.4 1420.96  4684.6 1425.36  5024.8 1429.36  5074.1 1430.26
#Mann= 3 , 0 , 0
       0     .03       0    2268    .035       0  2413.6     .03       0
Bank Sta=2268,2413.6
XS Rating Curve= 0 ,0
Exp/Cntr=0.3,0.1

Type RM Length L Ch R = 1 ,101890. ,485,485,485
BEGIN DESCRIPTION:
5000
END DESCRIPTION:
#Sta/Elev= 30
       0 1431.56    60.5 1430.96   527.5 1424.56   994.5 1420.96  1059.7 1420.66
  1461.5 1419.86  1928.5 1419.76  2053.3 1419.86  2103.7 1419.76  2132.9 1419.86
    2162 1420.56  2173.8 1420.06  2191.2 1418.96  2220.4 1417.26  2249.6 1414.26
  2270.6 1419.26  2278.8 1421.76    2308 1427.16  2319.1 1424.76  2337.2 1421.06
  2367.5 1419.26  2377.1 1419.16  2395.6 1418.26  2609.7 1419.16  3796.6 1419.46
  4159.7 1421.46  4263.6 1422.16  4730.6 1426.36  4934.7 1430.26    4982 1431.26
#Mann= 3 , 0 , 0
       0     .03       0    2162    .035       0    2308     .03       0
Bank Sta=2162,2308
XS Rating Curve= 0 ,0
Exp/Cntr=0.3,0.1

Type RM Length L Ch R = 1 ,101405. ,520,520,520
BEGIN DESCRIPTION:
4900
WEST:  Measured back 300 feet from zero to obtain 1428 ft elevation.  Added 300 feet contstant to all stations. (RCFCD photo maps)
END DESCRIPTION:
#Sta/Elev= 30
       0 1430.56     300 1426.36   369.3 1425.86   766.6 1422.16  1146.2 1420.86
  1233.2 1420.46  1699.8 1419.26    1923 1419.16  2166.4 1418.36  2437.6 1419.66
  2493.3 1419.36  2512.1 1419.46  2522.5 1419.76  2551.7 1420.96  2560.7 1420.06
  2580.8 1417.76    2610 1417.86  2639.1 1415.46  2657.8 1419.66  2668.3 1422.56
  2697.5 1425.06  2706.3 1423.16  2726.6 1419.86  3099.6 1419.06  3476.8 1418.66
  3566.3 1418.66  4253.6 1422.76  4499.5 1424.56  4966.1 1433.26  5067.4 1435.56
#Mann= 3 , 0 , 0
       0     .03       0  2551.7    .035       0  2697.5     .03       0
Bank Sta=2551.7,2697.5
XS Rating Curve= 0 ,0
Exp/Cntr=0.3,0.1

Type RM Length L Ch R = 1 ,100885. ,480,480,480
BEGIN DESCRIPTION:
4800
END DESCRIPTION:
#Sta/Elev= 30
       0 1432.26   281.9 1428.36   743.7 1423.86   748.1 1422.46  1522.3 1420.06
  1680.5 1419.36    2301 1418.96  2464.6 1419.06  2495.6 1418.96  2525.5 1419.16
  2544.3 1419.46  2554.7 1419.86  2583.8 1418.36  2592.9 1417.36  2641.6 1415.56
  2671.2 1418.16  2690.3 1423.66  2700.4 1426.16  2729.5 1423.46  2738.9 1422.06
  2758.6 1420.76  2783.7 1420.16  3079.2 1419.26  3079.6 1418.96  3545.4 1417.96
    4500 1422.56    4800 1426.56    4940 1430.56    5100 1434.56    5200 1438.56
#Mann= 3 , 0 , 0
       0     .03       0  2554.7    .035       0  2700.4     .03       0
Bank Sta=2554.7,2700.4
XS Rating Curve= 0 ,0
Exp/Cntr=0.3,0.1

Type RM Length L Ch R = 1 ,100405. ,505,505,505
BEGIN DESCRIPTION:
4700
WEST:  Measured 600 feet back from zero to obtain 1428 ft elevation.  Added 600 ft constant to all stations. (RCFCD photo maps)
END DESCRIPTION:
#Sta/Elev= 29
       0 1430.56     600 1426.36  1097.5 1422.26  1564.3 1419.46  1744.2 1419.26
  2497.8 1419.06  2520.3 1419.16    2702 1418.56  2714.3 1418.56  2731.1 1418.76
  2760.3 1419.26  2762.8 1419.36  2789.5 1418.46  2811.4 1416.16  2818.7 1415.96
  2847.8 1416.16 2859.96 1415.16    2877 1415.86  2906.2 1426.16  2908.4 1426.46
  2956.9 1420.86  2964.5 1420.46  3009.9 1419.96  3431.3 1418.46    4920 1422.56
    5200 1426.56    5340 1430.56    5540 1434.56    5700 1438.56
#Mann= 3 , 0 , 0
       0     .03       0  2762.8    .035       0  2908.4     .03       0
#XS Ineff= 2 , 0
       0    1656 1427.56               0
Permanent Ineff=
       F       F
Bank Sta=2762.8,2908.4
XS Rating Curve= 0 ,0
Exp/Cntr=0.3,0.1

Type RM Length L Ch R = 1 ,99900.  ,510,510,510
BEGIN DESCRIPTION:
4600
WEST:  Measured 310 feet back from zero to obtain 1428 ft elevation.  Added 310 constant to all stations. (RCFCD photo maps)
END DESCRIPTION:
#Sta/Elev= 30
       0 1430.56     310 1425.46   745.1 1422.96  1210.7 1419.86  1676.4 1418.86
    1757 1418.76    2142 1419.06  2538.3 1419.06  2607.7 1417.46  2640.7 1418.56
    2695 1418.46    2724 1418.86  2733.6 1419.46  2753.1 1420.26  2782.4 1415.96
  2811.4 1415.86  2831.3 1414.46  2840.5 1414.26  2869.6 1420.56  2880.1 1423.06
  2898.7 1424.66  2927.8 1418.56  2979.8 1418.16  3073.3 1418.16  3319.6 1417.26
    4310 1422.56    4590 1426.56    4810 1430.56    4990 1434.56    5210 1438.56
#Mann= 3 , 0 , 0
       0     .03       0  2753.1    .035       0  2898.7     .03       0
#XS Ineff= 2 , 0
       0    1902 1427.56               0
Permanent Ineff=
       F       F
Bank Sta=2753.1,2898.7
XS Rating Curve= 0 ,0
Exp/Cntr=0.3,0.1

Type RM Length L Ch R = 1 ,99390.  ,490,490,490
BEGIN DESCRIPTION:
4500
WEST:  Measure back 310 feet to obtain 1428 ft elevation.  Added 310 constant to all stations. (RCFCD photo maps)
END DESCRIPTION:
#Sta/Elev= 26
       0 1430.56     310 1426.36   456.8 1424.56  1029.7 1420.56  1389.8 1419.56
  1856.4 1419.26  2322.9 1419.16  2738.1 1418.76  2760.3 1418.86  2778.4 1420.16
  2789.5 1420.56  2818.6 1416.66  2847.8 1415.76  2875.6 1414.46    2877 1414.46
  2924.1 1424.76  2935.3 1425.36  2964.4 1418.56  2972.7 1418.46  3022.7 1418.26
  3051.9 1418.26  3072.4 1417.16    3256 1418.16    4310 1422.56    4510 1430.56
    4910 1438.56
#Mann= 3 , 0 , 0
       0     .03       0  2789.5    .035       0  2935.3     .03       0
#XS Ineff= 2 , 0
       0    2053 1427.56               0
Permanent Ineff=
       F       F
Bank Sta=2789.5,2935.3
XS Rating Curve= 0 ,0
Exp/Cntr=0.3,0.1

Type RM Length L Ch R = 1 ,98900.  ,510,510,510
BEGIN DESCRIPTION:
4400
WEST: Measured back 250 feet from zero to obtain 1428 contour interval.  Added 250 constant to all stations...
(RCFCD photo maps)
END DESCRIPTION:
#Sta/Elev= 29
       0 1430.56     250 1426.46   582.4 1423.86  1060.8 1422.26  1515.7 1419.36
  1837.4 1419.16  1982.4 1419.16  2449.1 1419.26    2614 1417.66    2677 1418.16
  2711.1 1418.16  2740.7 1418.06  2759.7 1418.26  2769.9 1418.96    2799 1417.06
  2808.2 1416.36  2828.2 1416.26  2856.7 1415.46  2857.4 1415.36  2886.5 1416.16
  2905.3 1423.06  2915.7 1425.86  2944.9 1418.66  2953.8 1418.06  3006.6 1418.16
    3850 1422.56    4350 1426.56    4490 1430.56    4650 1434.56
#Mann= 3 , 0 , 0
       0     .03       0  2769.9    .035       0  2915.7     .03       0
#XS Ineff= 2 , 0
       0    2254 1427.56               0
Permanent Ineff=
       F       F
Bank Sta=2769.9,2915.7
XS Rating Curve= 0 ,0
Exp/Cntr=0.3,0.1

Type RM Length L Ch R = 1 ,98390.  ,495,495,495
BEGIN DESCRIPTION:
4300
END DESCRIPTION:
#Sta/Elev= 30
       0 1432.06   161.9 1429.26     628 1423.66   680.8 1423.26    1094 1421.26
  1460.5 1420.56    1560 1420.16    2026 1419.06  2240.1 1418.96    2958 1418.96
  3019.7 1419.46  3062.6 1418.86  3117.2 1418.86  3161.9 1419.16  3165.9 1418.76
    3191 1415.26  3214.7 1414.56  3220.1 1414.26  3249.3 1415.46  3263.4 1419.06
  3278.4 1423.16  3307.5 1420.86  3312.1 1420.06  3336.6 1418.26  3384.7 1418.36
    3424 1419.46    4400 1422.56    4600 1426.56    4740 1430.56    4900 1434.56
#Mann= 3 , 0 , 0
       0     .03       0  3161.9    .035       0  3278.4     .03       0
Bank Sta=3161.9,3278.4
XS Rating Curve= 0 ,0
Exp/Cntr=0.3,0.1

Type RM Length L Ch R = 1 ,97895.  ,490,490,490
BEGIN DESCRIPTION:
4200
END DESCRIPTION:
#Sta/Elev= 30
       0 1430.96     422 1426.46   887.6 1421.36  1353.1 1420.56  1818.7 1418.66
  2284.2 1418.86  2749.8 1419.66  3164.4 1418.96  3182.5 1419.16  3213.2 1418.86
  3244.4 1418.96  3262.1 1419.26  3273.5 1419.06  3302.6 1415.96  3331.7 1413.76
  3359.8 1416.06  3360.8 1416.26  3389.9 1424.26  3408.7 1425.96    3419 1424.56
  3448.1 1419.06  3457.5 1418.66  3477.2 1418.46    3500 1418.76  3680.9 1418.86
  3946.2 1420.86    4200 1422.56    4360 1426.56    4600 1434.56    4700 1438.56
#Mann= 3 , 0 , 0
       0     .03       0  3262.1    .035       0  3408.7     .03       0
Bank Sta=3262.1,3408.7
XS Rating Curve= 0 ,0
Exp/Cntr=0.3,0.1

Type RM Length L Ch R = 1 ,97405.  ,510,510,510
BEGIN DESCRIPTION:
4100
END DESCRIPTION:
#Sta/Elev= 30
       0 1431.36   188.7 1428.66   654.3 1424.16   941.4 1421.86  1119.9 1420.56
  1585.4 1419.96    2051 1419.06  2516.6 1419.86  2982.2 1419.46  3286.4 1416.66
  3287.4 1418.66  3302.3 1418.76  3331.4 1418.76  3335.2 1418.86  3360.5 1419.06
  3389.6 1415.76  3418.7 1414.36  3432.9 1413.36  3447.8 1413.76  3476.9 1421.36
  3481.8 1422.56    3506 1425.46  3530.7 1419.66  3535.1 1418.86  3564.2 1418.26
  3598.3 1418.36  3913.3 1420.36    4068 1422.16  4378.9 1426.76  4736.9 1442.16
#Mann= 3 , 0 , 0
       0     .03       0  3360.5    .035       0    3506     .03       0
Bank Sta=3360.5,3506
XS Rating Curve= 0 ,0
Exp/Cntr=0.3,0.1

Type RM Length L Ch R = 1 ,96895.  ,495,495,495
BEGIN DESCRIPTION:
4000
END DESCRIPTION:
#Sta/Elev= 30
       0 1431.96   211.9 1427.96   325.5 1426.56   792.2 1421.36   988.3 1420.66
  1258.9 1419.96  1725.6 1415.76  1764.6 1415.96  2192.3 1419.26  2659.1 1419.36
  3125.8 1417.46  3299.1 1418.26  3317.3 1418.26  3329.9 1418.16  3359.1 1419.56
  3365.8 1419.06  3388.3 1416.26  3417.4 1413.96  3446.6 1413.26  3462.8 1416.46
  3475.8 1419.86    3505 1426.26  3511.3 1424.86  3534.1 1418.66  3559.9 1417.66
  3596.7 1418.06  4059.2 1420.46  4093.6 1421.66  4525.9 1440.86    4537 1441.46
#Mann= 3 , 0 , 0
       0     .03       0  3359.1    .035       0    3505     .03       0
Bank Sta=3359.1,3505
XS Rating Curve= 0 ,0
Exp/Cntr=0.3,0.1

Type RM Length L Ch R = 1 ,96400.  ,500,500,500
BEGIN DESCRIPTION:
3900
WEST:  Measured back 350 feet to obtain 1428 ft elevation.
Added 350 feet constant to all stations.
Measured 50 feet from station 3946.9 with an elevation of 1426 to obtain an elevation of 1428 (RCFCD photo maps)
END DESCRIPTION:
#Sta/Elev= 28
       0 1430.56     350 1424.76   611.2 1420.56   665.2 1420.36  1076.5 1419.56
  1448.3 1418.96  1541.8 1418.96    2007 1418.46  2231.3 1418.36  2472.3 1418.56
  2974.9 1418.16  2995.8 1418.36  3024.9 1419.16  3053.9 1417.06  3063.3 1415.86
    3083 1414.06  3112.3 1413.06  3141.2 1419.86  3161.2 1424.76  3170.3 1426.26
  3199.3 1419.86  3210.2 1418.56  3228.4 1417.76  3272.9 1417.96  3402.9 1417.96
  3797.5 1423.56  3868.2 1425.36  3996.9 1430.56
#Mann= 3 , 0 , 0
       0     .03       0  3024.9    .035       0  3170.3     .03       0
#XS Ineff= 2 , 0
       0     900 1422.56               0
Permanent Ineff=
       F       F
Bank Sta=3024.9,3170.3
XS Rating Curve= 0 ,0
Exp/Cntr=0.3,0.1

Type RM Length L Ch R = 1 ,95900.  ,505,505,505
BEGIN DESCRIPTION:
3800
END DESCRIPTION:
#Sta/Elev= 27
       0 1430.96     273 1420.46   661.7 1418.06   737.7 1420.26  1202.3 1418.96
  1447.8 1418.66  1666.9 1418.66  2131.6 1419.56    2234 1419.56  2596.2 1419.16
  2959.3 1417.86  2973.7 1417.76  3002.8 1418.66  3020.2 1418.06  3031.8 1417.16
  3060.8 1413.66  3069.3 1413.16  3089.9 1412.96  3118.9 1417.96    3148 1425.26
  3167.6 1423.66    3177 1421.56    3206 1417.36  3244.6 1417.66  3525.5 1418.56
  3665.9 1421.36    4120 1430.56
#Mann= 3 , 0 , 0
       0     .03       0  3002.8    .035       0    3148     .03       0
#XS Ineff= 2 , 0
       0    1250 1422.56               0
Permanent Ineff=
       F       F
Bank Sta=3002.8,3148
XS Rating Curve= 0 ,0
Exp/Cntr=0.3,0.1

Type RM Length L Ch R = 1 ,95395.  ,495,495,495
BEGIN DESCRIPTION:
3700
WEST:  Measured back 250 feet from zero to obtain 1428 ft elevation.  Added 250 constant to all stations.  Added station 170 for elevation 1424 (RCFCD photo maps)
END DESCRIPTION:
#Sta/Elev= 29
       0 1430.56     170 1426.56     250 1424.66   622.4 1421.26   949.2 1421.26
  1088.6 1422.06  1554.8 1419.66  1727.9 1421.06    2021 1419.56  2506.7 1418.96
  2953.4 1418.16  3174.9 1416.56  3188.1 1416.86  3215.6 1418.36  3236.8 1418.96
  3244.7 1418.76  3273.9 1414.66  3285.5 1413.46    3303 1412.46  3332.2 1416.06
  3361.3 1421.96  3382.8 1425.46  3390.4 1425.56  3419.6 1418.46  3431.5 1417.96
  3448.7 1417.66  3483.7 1417.86  3885.8 1422.36  4097.7 1431.86
#Mann= 3 , 0 , 0
       0     .03       0  3236.8    .035       0  3390.4     .03       0
#XS Ineff= 2 , 0
       0    1600 1422.56               0
Permanent Ineff=
       F       F
Bank Sta=3236.8,3390.4
XS Rating Curve= 0 ,0
Exp/Cntr=0.3,0.1

Type RM Length L Ch R = 1 ,94900.  ,500,500,500
BEGIN DESCRIPTION:
3600
END DESCRIPTION:
#Sta/Elev= 29
       0 1426.56     240 1422.56     260 1424.46   665.4 1421.26   890.7 1418.96
  1131.5 1418.26  1597.7 1418.16  1669.5 1418.26  2530.1 1418.66  2996.3 1418.16
  3075.6 1416.46  3083.6 1415.56  3112.8 1415.56  3129.8 1417.86  3141.9 1419.16
    3171 1417.46  3200.2 1413.36  3227.2 1413.36  3229.3 1413.56  3258.5 1419.76
  3275.8 1424.46  3287.6 1426.36  3316.7 1419.66  3324.5 1418.96  3345.9 1417.96
  3378.3 1417.56  3462.4 1418.06  3928.6 1430.26  4035.4 1435.06
#Mann= 3 , 0 , 0
       0     .03       0  3141.9    .035       0  3287.6     .03       0
#XS Ineff= 2 , 0
       0    1900 1422.56               0
Permanent Ineff=
       F       F
Bank Sta=3141.9,3287.6
XS Rating Curve= 0 ,0
Exp/Cntr=0.3,0.1

Type RM Length L Ch R = 1 ,94400   ,480,480,480
BEGIN DESCRIPTION:
3500
END DESCRIPTION:
#Sta/Elev= 30
       0 1428.06   200.5 1425.16   415.1 1422.86   882.1 1419.26   975.6 1418.86
  1349.1 1418.06  1750.8 1417.66  1816.1 1417.76    2283 1419.26  2525.9 1419.56
    2750 1425.26  3163.8 1416.26  3187.9 1417.76  3204.2 1416.06  3217.1 1414.36
  3246.2 1415.36  3252.6 1415.26  3275.4 1413.26  3301.1 1412.76  3304.6 1413.06
  3333.8 1419.16  3349.5 1423.16    3363 1424.36  3392.2 1417.56    3398 1417.26
  3421.3 1417.16  3450.8 1417.06    3684 1419.86  4076.2 1426.16  4131.1 1432.86
#Mann= 3 , 0 , 0
       0     .03       0  3252.6    .035       0  3333.8     .03       0
#XS Ineff= 2 , 0
       0    2800 1422.56    3800       0 1422.56
Permanent Ineff=
       F       F
Bank Sta=3252.6,3333.8
XS Rating Curve= 0 ,0
Exp/Cntr=0.3,0.1
